HEC-RAS study HECRAS_v1.prj: HECRAS_v1

--- HECRAS_v1.g01 (geometry) --- (continued)

Type RM Length L Ch R = 1 ,3866.315,225.37,200,174.75
XS GIS Cut Line= 4
    1080660.7755    1570590.9984    1080958.4221    1570667.3234
    1081175.4436    1570853.3408    1081659.8275    1571156.3035
#Sta/Elev= 30
       0   77.02  108.83    77.5  231.58    77.7  313.44      78  335.73      78
  362.24    77.5  374.15      77  396.85    76.5  403.98      76  414.38      75
  440.59      75  443.95    75.5  451.88   76.99  455.46    77.5  458.75    77.5
  491.12    77.5  523.92   77.65  547.04    77.5   575.5   77.61  606.89   78.01
   648.6   78.24  736.29   78.61  781.16   78.69  819.96   78.92  841.68   78.93
  884.92   79.19 1003.74   79.49 1047.54   79.36 1109.03   78.86 1164.44   78.91
#Mann= 3 ,0,0
       0    .035       0  362.24    .018       0  458.75    .035       0
Bank Sta=362.24,458.75
XS Rating Curve= 0 ,0
Exp/Cntr=0.3,0.1

Type RM Length L Ch R = 1 ,3666.315,208.53,200,191.35
XS GIS Cut Line= 4
    1080591.5109    1570888.9546    1080787.6296    1570935.8453
     1081141.525    1570888.6593    1081641.6243    1571220.7033
#Sta/Elev= 30
       0   76.87    25.8      77  214.53      77  277.74   77.15  314.23   77.31
  335.05    77.5  353.25    77.5  362.73      77  365.18    76.5  373.23    74.5
  390.54    74.5  398.08      75  404.18    75.5   414.4    76.5  421.85      77
  491.43    77.5  620.24    77.5  668.23   77.92  719.59      78  751.47    78.4
  758.02   78.39  771.36   78.18  788.12   78.16  804.82   78.25   823.6    78.5
  872.58   78.62  947.16   78.97 1010.47   78.79 1063.58   78.26 1158.97   78.17
#Mann= 3 ,0,0
       0    .035       0  353.25    .018       0  491.43    .035       0
Bank Sta=353.25,491.43
XS Rating Curve= 0 ,0
Exp/Cntr=0.3,0.1

Type RM Length L Ch R = 1 ,3466.315,196.37,200,203.63
XS GIS Cut Line= 4
     1080606.752    1571080.9971    1080921.7505    1571143.2625
    1081221.8512    1571010.8655    1081624.2068    1571282.5043
#Sta/Elev= 30
       0   75.86   114.1   76.03  215.51    76.5  319.04   76.74  366.74      77
  471.31      77  473.26      77  478.48    76.5   489.7    74.5  494.18      74
  509.17      74  514.75    74.5  522.46      76  525.79    76.5  531.31    76.8
  535.57      77  584.65      77  607.19    77.5  734.46    77.5  764.18   77.71
  801.81   77.78  826.78   78.04  897.13   78.31  957.89   78.16  994.73   77.81
  1012.4   77.74 1050.79   77.73 1083.48   77.51 1112.89   77.19 1134.57   77.17
#Mann= 3 ,0,0
       0    .035       0  471.31    .018       0  531.31    .035       0
Bank Sta=471.31,531.31
XS Rating Curve= 0 ,0
Exp/Cntr=0.3,0.1

Type RM Length L Ch R = 1 ,3266.315,184.79,200,215.21
XS GIS Cut Line= 4
    1080595.0101    1571256.4086    1080957.9986    1571317.8097
    1081316.1518    1571209.0849    1081593.8293    1571399.4434
#Sta/Elev= 30
       0    75.5  100.87   75.51  180.22      76  215.05      76  308.54    76.5
   343.4    76.5  430.16      77  495.72      77  506.44   76.49  511.56   76.37
  534.21   76.35  547.17   76.18  551.66      76  563.52    74.5  568.16      74
  574.91    73.5  583.66    73.5  589.15      74  600.69      76  607.17   77.01
  632.77   77.33  665.46      77  899.52   77.01  950.09   76.84   992.1    76.5
 1002.96    76.5 1027.01      76 1044.84      75 1065.64      76  1079.1   76.25
#Mann= 3 ,0,0
       0    .035       0  547.17    .018       0  607.17    .035       0
Bank Sta=547.17,607.17
XS Rating Curve= 0 ,0
Exp/Cntr=0.3,0.1

Type RM Length L Ch R = 1 ,3066.315,165.67,200,234.33
XS GIS Cut Line= 4
    1080510.4142    1571327.4268    1080932.1897    1571407.2786
    1081343.4433    1571495.4044    1081546.3129    1571648.9608
#Sta/Elev= 30
       0    75.5  141.84    75.5  249.87      76  300.64      76  375.41    76.5
  396.52    76.5  492.71      77  524.68      77  564.84    76.5  575.39   75.99
  589.07    75.5  622.19   75.07  632.03      75   648.1    73.5  654.41    73.5
  661.02      74  668.93      75   679.2    76.5  682.19   76.53  732.44   76.72
  771.91    76.5   841.3   76.38  889.54      76  932.18    75.5  947.53    74.5
  952.91    74.9  958.64    75.5 1029.37   75.76  1055.2      76 1104.29      76
#Mann= 3 ,0,0
       0    .035       0  622.19    .018       0  682.19    .035       0
Bank Sta=622.19,682.19
XS Rating Curve= 0 ,0
Exp/Cntr=0.3,0.1

Type RM Length L Ch R = 1 ,2866.315,192.19,200,207.81
XS GIS Cut Line= 4
    1080480.4185    1571356.0345    1080998.9119    1571452.4209
    1081074.7051    1571789.2748    1081372.5527    1572002.1389
#Sta/Elev= 30
       0    75.5  155.77    75.5  263.17      76  314.66      76  394.08    76.5
  509.81      77  540.56      77  597.49    76.5   628.7      76  636.94      76
  642.91   75.78  650.75    75.5  670.45    73.5  693.83    73.5  702.91   74.75
  711.22      76  721.63    76.5  737.08    76.5  798.69      76   880.5    75.5
  895.95   74.64   915.7   74.17   927.3    73.5  936.17    73.5  940.58      74
  947.45      75  952.29    75.5 1070.23    75.5 1101.31   75.63 1238.74   75.79
#Mann= 3 ,0,0
       0    .035       0  642.91    .018       0  702.91    .035       0
Bank Sta=642.91,702.91
XS Rating Curve= 0 ,0
Exp/Cntr=0.3,0.1

Type RM Length L Ch R = 1 ,2666.315,198.69,200,201.31
XS GIS Cut Line= 4
    1080413.8089    1571417.1216    1080837.3071    1571491.9031
     1080825.417    1571801.0496    1081227.9039    1572100.2957
#Sta/Elev= 30
       0    75.3   59.54    75.5  118.93    75.5  229.11      76  290.18      76
  416.93    76.5  490.59    76.5  509.01      76   519.1   75.45  530.54    74.5
  538.59   73.51  546.13      73  559.12      73  573.11   73.99   579.1    74.3
  591.04      75  600.21      76  609.19    76.5  623.05    76.5  680.09      76
   693.4      76  760.36    75.5  900.59    75.5  950.83      75  962.64    73.5
  968.92    73.5  981.86      75 1099.24   75.18 1187.19   75.13 1240.97   75.31
#Mann= 3 ,0,0
       0    .035       0   519.1    .018       0   579.1    .035       0
Bank Sta=519.1,579.1
XS Rating Curve= 0 ,0
Exp/Cntr=0.3,0.1

Type RM Length L Ch R = 1 ,2466.315,249.51,200,150.31
XS GIS Cut Line= 4
    1080356.2232    1571464.6942    1080655.8705    1571508.8005
    1080636.4999    1571737.3738    1081190.6132    1572157.6623
#Sta/Elev= 27
       0   75.05  231.45      76  414.03      76  417.14   75.93  419.77   75.73
  426.04      75  436.16    73.5  440.94      73  447.68    72.5   458.7    72.5
  466.35    73.5  468.97      74  475.54    75.5  478.49      76  479.77   76.06
  488.87   76.42  512.11   76.42  681.57   75.57  783.39   75.34  887.13    75.3
   925.6      75  931.26    74.5  935.05      74   945.2      74  953.65      75
 1152.64      75 1227.74    75.3
#Mann= 3 ,0,0
       0    .035       0  419.77    .018       0  479.77    .035       0
Bank Sta=419.77,479.77
XS Rating Curve= 0 ,0
Exp/Cntr=0.3,0.1

Type RM Length L Ch R = 1 ,2266.315,208.24,200,191.76
XS GIS Cut Line= 4
    1080212.2983    1571692.6391    1080255.2301    1571702.1731
    1080547.5626    1571712.6135     1081148.028    1572190.0326
#Sta/Elev= 30
       0   74.88  134.68    75.5  194.08      76  222.74      76  224.25   75.87
  228.63    75.5  235.47      74  238.21    73.5  242.68      73  248.74   72.62
  257.67   72.69     266      73  273.15    73.5  284.25   74.45  294.88    75.5
  308.28   75.97  341.67      76  376.61   76.24  473.47   76.08  559.15    75.5
  603.46    75.5  780.73      75  800.12    74.5  815.02    73.5  821.27    73.5
  834.08      75  926.94   74.91  932.61      75 1021.16      75 1103.63   75.29
#Mann= 3 ,0,0
       0    .035       0  224.25    .018       0  284.25    .035       0
Bank Sta=224.25,284.25
XS Rating Curve= 0 ,0
Exp/Cntr=0.3,0.1

Type RM Length L Ch R = 1 ,2066.315,211.93,200,188.07
XS GIS Cut Line= 4
    1080078.1307    1571881.4182    1080317.4153     1571947.621
    1080645.3778    1571866.6952    1081111.3766    1572231.5927
#Sta/Elev= 30
       0   74.52   211.7      75  300.93    75.5  391.45    75.5  395.62    75.5
  401.35      75   414.2      73  420.87    72.5  428.26    72.5  435.78      73
  444.61    74.5  451.45    75.2   455.9    75.5  509.59      76  564.57      76
  638.95    75.5  861.11      75  865.39    74.5  870.63    73.5  879.49   73.01
   883.8   73.32  891.84    74.5   897.7      75  951.24      75  966.65    74.5
  973.92    74.5  1003.7   74.96 1055.17      75 1127.79   75.46 1177.94    75.5
#Mann= 3 ,0,0
       0    .035       0  391.45    .018       0  451.45    .035       0
Bank Sta=391.45,451.45
XS Rating Curve= 0 ,0
Exp/Cntr=0.3,0.1

Type RM Length L Ch R = 1 ,1866.315,158.12,200,241.88
XS GIS Cut Line= 4
    1080035.6115    1571945.0255    1080541.2594    1572105.8958
    1080680.2679    1572002.6317    1081065.8008    1572304.3412
#Sta/Elev= 30
       0    74.5   72.07   74.54  205.82      75  217.69    75.5   230.6    75.5
  250.24      75  258.43      75  280.63    75.5  370.62    75.5  446.42      76
  476.36      76  555.16    75.5  559.14    75.5  564.22      75  574.28      73
  580.04    72.5  601.97    72.5  606.75      73  615.16   74.42  624.78   75.57
  720.12    75.5  796.96   75.02  840.82   74.57  871.58    74.5  875.56      74
  883.22    72.5  891.13    72.5  914.23    74.5 1081.66   74.84 1193.34   75.47
#Mann= 3 ,0,0
       0    .035       0  555.16    .018       0  615.16    .035       0
Bank Sta=555.16,615.16
XS Rating Curve= 0 ,0
Exp/Cntr=0.3,0.1

Type RM Length L Ch R = 1 ,1666.315,177.66,200,222.34
XS GIS Cut Line= 4
    1079970.6561    1571994.2082    1080329.7154    1572077.9904
    1080643.9976    1572369.1636    1080877.7629    1572548.1553
#Sta/Elev= 30
       0    74.5  229.07      75  309.06      75  317.96    75.2   368.7   75.47
  438.64    75.5  473.27      76  489.48      76  535.71    75.5  550.97    75.5
  556.53      75   567.8    72.5  572.23      72  577.77      72  590.06    72.5
   594.4      73  607.86      75  610.97   75.15  617.83    75.5  629.63    75.5
  735.03    74.5  797.14   74.21  940.89   73.87  991.57      74 1005.53    73.5
 1012.74    72.5 1022.07    72.5 1028.71    73.5  1033.1      74 1091.56      74
#Mann= 3 ,0,0
       0    .035       0  550.97    .018       0  610.97    .035       0
Bank Sta=550.97,610.97
XS Rating Curve= 0 ,0
Exp/Cntr=0.3,0.1

Type RM Length L Ch R = 1 ,1466.315,215.04,200,184.95
XS GIS Cut Line= 4
    1079900.4549     1572041.573    1080314.2202    1572157.3594
    1080340.1248     1572473.396    1080710.0367    1572753.1583
#Sta/Elev= 30
       0    74.5   62.68    74.5  145.72   74.84   234.9      75  347.09      75
  442.19   75.47   490.9    75.5  553.27    74.5  568.45   74.03  573.79   73.79
  580.24   73.51  586.69      73  593.86      72  610.69      72  616.73    72.5
  627.34      74  633.83   74.83  635.08      75  652.52      75  750.56    74.5
  763.97    74.5  883.71      74  909.99      74 1032.79    73.5 1159.98    73.5
  1169.9      72 1175.51   72.01 1184.89    72.5 1194.77    73.5 1210.55    73.5
#Mann= 3 ,0,0
       0    .035       0  573.79    .018       0  633.83    .035       0
Bank Sta=573.79,633.83
XS Rating Curve= 0 ,0
Exp/Cntr=0.3,0.1

Type RM Length L Ch R = 1 ,1266.315,410.51,400,389.53
XS GIS Cut Line= 4
    1079784.3397     1572071.356    1080040.1108    1572163.4889
    1080243.6466    1572472.3018    1080683.0551    1572807.7735
#Sta/Elev= 30
       0   74.33   55.54    74.5   208.2    74.5  258.96      75  311.83      75
  375.49    75.5  418.48   75.43   431.8   75.26  440.92      75  446.31      74
  453.08   72.48  455.92      72  460.55    71.5  467.82    71.5  474.04      72
  477.82    72.5  486.19      74  489.47    74.5   491.8   74.69  496.21      75
   619.2      75  719.46    74.5  973.75    73.5 1165.84    73.5 1173.76      73
 1178.08    72.5 1182.58   72.19  1187.1      72 1188.63    72.1 1194.54    72.8
#Mann= 3 ,0,0
       0    .035       0   431.8    .018       0   491.8    .035       0
Bank Sta=431.8,491.8
XS Rating Curve= 0 ,0
Exp/Cntr=0.3,0.1

Type RM Length L Ch R = 1 ,866.3152,209.16,200,190.8
XS GIS Cut Line= 3
    1079643.4541    1572112.7012    1080005.4348    1572386.9289
    1080630.2867    1572854.0753
#Sta/Elev= 30
       0      74   43.11      74   63.48   74.12  151.63      74  180.83    74.5
  219.59    74.5  222.51    74.5  227.04      74  237.66      72  241.66    71.5
  261.73    71.5  268.17    72.5  275.29      74  279.23    74.5     280    74.5
  350.02    74.5  378.36   74.64  423.61    74.5  435.04   74.65  486.71    74.5
  555.69    74.5  604.18   74.74  630.84      75  703.11      75  785.12    74.5
  859.83   74.27  997.67    73.5 1047.47    73.5 1194.82   73.13  1234.3   73.43
#Mann= 3 ,0,0
       0    .035       0  219.59    .018       0     280    .035       0
Bank Sta=219.59,280
XS Rating Curve= 0 ,0
Exp/Cntr=0.3,0.1

Type RM Length L Ch R = 1 ,666.3153,201.09,200,198.91
XS GIS Cut Line= 3
     1079545.912    1572344.5175     1079874.612    1572461.9099
    1080500.4923    1572908.3154
#Sta/Elev= 25
       0   73.68  138.79   74.49  141.01    74.5  148.27      74  151.99    73.5
  160.17    71.5  162.81      71  177.32      71  181.77   71.63  191.54    73.5
  195.51      74  198.79      74  273.97   74.16  307.62      74   437.4      74
  477.62   74.35  524.23    74.5   577.9    74.5  601.32   74.35  642.99    74.5
  840.62    74.5  848.79   74.71  862.69    74.5  935.95   74.49  1117.8   73.26
#Mann= 3 ,0,0
       0    .035       0  138.79    .018       0  198.79    .035       0
Bank Sta=138.79,198.79
XS Rating Curve= 0 ,0
Exp/Cntr=0.3,0.1

Type RM Length L Ch R = 1 ,466.3153,133.35,138.85,144.35
XS GIS Cut Line= 3
    1079485.0302    1572529.6118     1079885.609      1572655.92
    1080224.8188    1572885.3892
#Sta/Elev= 26
       0   73.45   48.82    73.5  148.09      74  188.66      74  195.95   73.58
  202.63      73  212.77    71.5  219.46      71  227.92      71  235.69    71.5
  244.38      73  248.04    73.5  253.15      74  255.95      74  316.28      74
  376.01    73.5  459.96    73.5   487.3   73.85  504.04   73.95  550.53    73.5
  599.18   73.42  634.57    73.5  736.13    73.5  792.18   74.18  816.37   74.27
  829.56   74.21
#Mann= 3 ,0,0
       0    .035       0  195.95    .018       0  255.95    .035       0
Bank Sta=195.95,255.95
XS Rating Curve= 0 ,0
Exp/Cntr=0.3,0.1

Type RM Length L Ch R = 1 ,327.4682,124.13,327.54,124.31
XS GIS Cut Line= 3
    1079445.6949    1572613.6877    1079779.4184    1572790.7109
    1080103.7223    1572902.2829
#Sta/Elev= 20
       0   73.19   44.14    73.5  158.42    73.5  167.56    73.5   172.2      73
  181.88      71  187.32    70.5  190.49    70.5  198.68      71   208.4      72
  218.41   73.44   219.8   73.58  224.86      74  243.01      74  357.09    73.5
     382    73.5  471.16   73.18  549.23      73  668.41   73.04  720.73   73.49
#Mann= 3 ,0,0
       0    .035       0  158.42    .018       0   219.8    .035       0
Bank Sta=158.42,219.8
XS Rating Curve= 0 ,0
Exp/Cntr=0.3,0.1

River Reach=ARROYOELZORRO   ,ABAJOLAT1
Reach XY= 30
1079526.957286981573013.08491518    1079327.7203    1573037.6709
    1078910.1353    1572733.9715    1078253.1058    1572618.3051
    1078094.2524    1572733.3828     1077901.525    1572656.1992
    1077773.5463    1572795.8368    1077590.4555    1572744.3908
    1077195.6486    1573072.3463    1076992.2968    1573064.6889
    1076912.2578    1573236.1591    1076722.9953    1573202.6476
    1076612.4146    1573358.3916    1076411.5354    1573301.7432
     1076266.837    1573437.2883    1076101.9001    1573337.8544
    1075934.8719    1573443.2967    1075776.3981    1573325.9612
    1075314.2113    1573352.5123    1075021.8357    1573164.1616
    1074762.1036    1573307.0204    1074809.0672    1573474.3696
     1074606.396     1573339.961    1074520.4062    1573461.8019
    1074456.1675    1573323.7608    1074343.8516    1573398.9026
    1074180.2065    1573289.1003     1074305.487    1573190.8074
    1074104.9324     1572975.833    1073782.6483    1573130.3062

Type RM Length L Ch R = 1 ,8685.184,132.08,96,60.24
XS GIS Cut Line= 5
    1079689.4749    1572775.0158    1079573.3755    1572915.1394
    1079527.1627    1573013.1873     1079441.341    1573198.8588
    1079203.8048    1573913.9964
#Sta/Elev= 30
       0    73.7   68.38    73.5  207.45    73.5  240.31   71.24  249.34   71.24
  270.65   69.77  310.66   69.77  331.47   71.24  449.51   71.24  477.54   73.24
   510.5      73  597.78      73  699.99   72.01  722.46    70.5  739.33   70.27
  755.91    69.5  764.56    69.5  768.83      70  780.68      72  788.11    72.6
  802.42   72.93  815.94   72.83  827.78      73  856.22    71.5  863.31    71.5
  918.75    73.5  989.86    76.5 1031.74   77.47 1158.17    78.5 1248.47   78.74
#Mann= 3 ,0,0
       0    .035       0  249.34    .018       0  331.47    .035       0
Levee=-1,207.6,73.5,-1,477.97,73.24,	341,	340
Bank Sta=249.34,331.47
XS Rating Curve= 0 ,0
Exp/Cntr=0.3,0.1

Type RM Length L Ch R = 1 ,8589.181,71.26,107.16,143.04
XS GIS Cut Line= 5
    1079531.8761    1572688.6196    1079402.7592    1572950.0285
    1079453.2203    1573057.3448    1079460.9676    1573080.2037
    1079160.4004    1573894.0637
#Sta/Elev= 30
       0    73.5  212.39    73.5  246.26   71.08  328.15   71.11  349.15   69.68
  389.15   69.68  410.15   71.18  504.98   71.21  535.47   73.38  575.11      73
  669.62      73  708.06    72.5  721.73   71.19  730.62    70.5  744.79   70.14
  757.94    69.5  780.38    69.5  790.23   69.83  795.63   70.22  810.78   71.99
  817.23    72.5  879.82   72.37   890.5   72.16  906.69    71.5  927.06    71.5
  985.34   73.21 1044.39      76 1076.42   76.89 1227.07   78.49 1301.87    78.5
#Mann= 3 ,0,0
       0    .035       0  328.15    .018       0  410.15    .035       0
Levee=-1,211.38,73.5,-1,535.71,73.38,	341,	340
Bank Sta=328.15,410.15
XS Rating Curve= 0 ,0
Exp/Cntr=0.3,0.1

Type RM Length L Ch R = 1 ,8482.02 ,74.63,111.47,148.33
XS GIS Cut Line= 4
    1079486.3677    1572661.6321    1079419.3723    1572857.7406
    1079292.7963    1573129.7306    1079063.1393    1573850.2486
#Sta/Elev= 30
       0    73.5  218.95   73.46  252.64   71.05  367.49   71.05  388.54   69.58
  428.82   69.58  449.82   71.05  461.84   71.05  495.23   73.48  503.71    73.5
  511.53      73  525.43    70.5  534.64    69.5  571.54    69.5  577.94      70
  594.06    72.5   605.9   73.31  636.65      73  759.24      73  764.93    72.5
  775.55    70.5  782.78    69.5  796.46    69.5  827.74      72  869.52   71.79
  888.29      71  901.54      71 1081.42    76.5 1203.96      78 1263.47   78.16
#Mann= 3 ,0,0
       0    .035       0  367.49    .018       0  449.82    .035       0
Levee=-1,219.27,73.5,-1,495.44,73.49,	341,	340
Bank Sta=367.49,449.82
XS Rating Curve= 0 ,0
Exp/Cntr=0.3,0.1

Type RM Length L Ch R = 1 ,8370.554,128.33,91.45,54.52
XS GIS Cut Line= 6
    1079448.3734    1572649.6729    1079387.8709    1572843.0808
    1079344.2332    1572935.8468    1079236.2393    1572961.8225
     1079212.153    1572968.0202    1078982.7058    1573824.8486
#Sta/Elev= 30
       0   73.22   33.56   73.11  216.39   73.27  248.05   71.01  334.24   70.98
  355.24   69.48  395.24   69.48  416.24   70.91  509.33    70.9  537.96   72.92
  548.92      73  642.28   72.98  768.63    72.5  924.21    72.5  942.88      71
  954.78    69.5  963.72    69.5   971.2   69.18  980.22    69.5  986.24   70.17
  995.65    71.5 1003.15      72 1024.17   72.34 1039.11   72.73 1068.18    73.9
 1090.81    74.5 1137.54      76 1183.97      77 1309.43      78 1328.13   78.03
#Mann= 3 ,0,0
       0    .035       0  334.24    .018       0  416.24    .035       0
Levee=-1,216.11,73.27,-1,549.07,73.01,	341,	340
Bank Sta=334.24,416.24
XS Rating Curve= 0 ,0
Exp/Cntr=0.3,0.1

Type RM Length L Ch R = 1 ,8279.103,143.28,107.05,70.86
XS GIS Cut Line= 4
    1079359.4733    1572590.4061    1079272.7216    1572789.4938
    1079146.1456    1573061.4837    1078894.6523    1573793.5218
#Sta/Elev= 30
       0      73  124.03      73  236.91    72.7  262.57   70.86  270.55   70.86
  291.77   69.39  331.85    69.4  353.22   70.86  471.77   70.86  496.41   72.62
  515.77   72.68  600.11   72.76  788.72   72.12  939.38    72.5  958.72      72
  977.18    70.5  995.44    70.5 1008.04      70 1014.04    69.5  1024.6      69
 1036.88      69 1041.74   69.49 1056.77   71.46 1070.54    73.5 1078.59      74
 1092.19    74.5  1145.6      76 1225.16    77.5 1269.15      78  1291.2      78
#Mann= 3 ,0,0
       0    .035       0  270.55    .018       0  353.22    .035       0
Levee=-1,236.62,72.7,-1,496.9,72.62,	341,	340
Bank Sta=270.55,353.22
XS Rating Curve= 0 ,0
Exp/Cntr=0.3,0.1

Type RM Length L Ch R = 1 ,8172.052,72.42,108.66,144.91
XS GIS Cut Line= 6
    1079236.8122    1572529.6153    1079140.6199    1572728.0176
    1079096.0536    1572807.9575    1079149.5197     1572919.071
     1079160.612    1572940.2495    1078827.2364    1573784.8012
#Sta/Elev= 30
       0      73   60.19      73  129.66   72.54  240.63    72.5  266.01   70.69
  353.32   70.72  374.32   69.29  414.32   69.29  435.32   70.79  529.97   70.82
  553.46    72.5   631.7   72.63  725.27    72.5  844.52      72  984.55      72
 1014.89    72.4 1040.75      72 1070.66      71 1079.68    70.5 1107.13      70
 1116.99      69 1134.46      69  1138.6    69.5 1140.93      70  1151.6   73.25
 1159.01      74 1253.53   76.49 1306.77      77 1352.23      78  1367.2      78
#Mann= 3 ,0,0
       0    .035       0  353.32    .018       0  435.32    .035       0
Levee=-1,239.77,72.51,-1,631.77,72.63,	341,	340
Bank Sta=353.32,435.32
XS Rating Curve= 0 ,0
Exp/Cntr=0.3,0.1

Type RM Length L Ch R = 1 ,8063.394,75.89,111.57,147.24
XS GIS Cut Line= 4
    1079207.1788    1572509.5069    1079114.7195    1572715.9643
    1078988.1435    1572987.9543    1078734.1028    1573749.8761
#Sta/Elev= 30
       0      73   63.41    72.5  245.85    72.5  271.62   70.66  388.31   70.66
  409.19   69.19  449.23   69.19  470.35   70.66  480.82   70.66  501.82   72.16
  526.22   72.16  526.96   71.91  687.74      72  756.24   71.72 1014.35      72
 1024.78      71 1037.96      69 1045.76    68.5 1051.26    68.5 1060.57      69
 1094.21      72 1105.86      72 1118.71      71  1133.7   70.96 1159.07   71.82
  1185.9    73.5  1222.2      75 1243.25   75.26 1282.31    76.3 1329.37   76.96
#Mann= 3 ,0,0
       0    .035       0  388.31    .018       0  470.35    .035       0
Levee=-1,246.08,72.51,-1,501.81,72.15994,	341,	340
Bank Sta=388.31,470.35
XS Rating Curve= 0 ,0
Exp/Cntr=0.3,0.1

Type RM Length L Ch R = 1 ,7951.827,132.49,93.75,55.01
XS GIS Cut Line= 6
    1079179.6621    1572494.6902    1079087.3428     1572703.224
    1079045.2535    1572789.9658    1078932.8887    1572820.4592
    1078914.0199    1572841.8243    1078634.6193     1573714.951
#Sta/Elev= 30
       0   72.91   47.57    72.5  247.93   72.45  273.46   70.62   358.9   70.59
   379.9   69.09   419.9   69.09   440.9   70.52  528.14   70.51   549.2   72.01
  573.68   72.02  575.23    71.5  694.23   71.71  826.92   71.31  1021.3   71.69
 1059.14   71.22 1110.43   71.93 1154.79      72 1178.52    71.5 1206.48   70.13
 1231.08   70.64 1280.53    68.5 1295.36    68.5 1308.85      69 1325.22    68.5
 1333.96      69 1342.84      70 1364.31   73.54 1374.45   74.56 1386.14      75
#Mann= 3 ,0,0
       0    .035       0   358.9    .018       0   440.9    .035       0
Levee=-1,247.66,72.45,-1,572.62,72.02,	341,	340
Bank Sta=358.9,440.9
XS Rating Curve= 0 ,0
Exp/Cntr=0.3,0.1

Type RM Length L Ch R = 1 ,7858.077,133.73,95.13,56.53
XS GIS Cut Line= 4
    1079064.8327    1572431.4018    1078954.4105    1572645.2909
    1078864.4802    1572883.4531     1078573.765     1573693.996
#Sta/Elev= 30
       0      73   28.62      73  102.49    72.5  122.09    72.5  150.87      72
  234.28   71.86  266.96   71.97  287.96   70.47  298.06   70.47  319.05      69
  359.06      69  380.13   70.47  497.16   70.47  518.16   71.97  542.56   71.97
  543.98    71.5  717.22    71.5  787.06   71.12  911.27    71.5 1078.53    71.5
 1193.12    71.9 1247.99   71.81 1272.48    71.5 1280.85    70.5 1293.84    69.5
 1316.32   68.71 1324.62   68.83 1335.22   69.37  1348.5      71 1356.39   71.61
#Mann= 3 ,0,0
       0    .035       0  298.06    .018       0  380.13    .035       0
Levee=-1,267.02,71.96504,-1,518.24,71.9697,	341,	340
Bank Sta=298.06,380.13
XS Rating Curve= 0 ,0
Exp/Cntr=0.3,0.1

Type RM Length L Ch R = 1 ,7762.949,78.48,114.34,150.19
XS GIS Cut Line= 6
    1078881.4231    1572348.1108    1078808.8085    1572598.7291
    1078784.9029    1572683.3915    1078852.9902    1572787.2213
    1078860.2564    1572814.6251    1078534.2891    1573687.5401
#Sta/Elev= 30
       0   72.58   62.27   72.53  120.78      72   260.3   71.62  260.85   71.81
  285.25   71.81  306.25   70.31  391.06   70.34  412.06   68.91  452.06   68.91
  473.06   70.41  566.41   70.43  587.41   71.93  611.82   71.93  613.12    71.5
  760.06    71.5  789.68   71.43  846.17      71 1039.93   71.46 1137.27   71.41
 1268.84   71.58 1358.38    71.5 1366.04      71 1373.51    69.5 1376.66      69
 1381.93    68.5 1399.68    68.5 1415.51    69.5 1430.31      70  1433.2   70.38
#Mann= 3 ,0,0
       0    .035       0  391.06    .018       0  473.06    .035       0
Levee=-1,285.33,71.8001,-1,587.45,71.9343,	341,	340
Bank Sta=391.06,473.06
XS Rating Curve= 0 ,0
Exp/Cntr=0.3,0.1

Type RM Length L Ch R = 1 ,7648.612,69.71,104.17,138.64
XS GIS Cut Line= 4
    1078856.8697    1572329.4841    1078785.7915    1572590.9508
    1078698.8347    1572878.1138    1078462.3223    1573660.4468
#Sta/Elev= 24
       0    72.5   78.19    72.5  138.34      72   270.9   71.56  271.41   71.56
  272.06   71.78  296.47   71.78  317.48   70.28  435.19   70.27  456.24    68.8
  496.27    68.8  517.26   70.27  526.77   70.27  547.78   71.77  572.19   71.77
  573.73   71.25  614.48   71.37  655.31   71.39   765.3      71 1194.14      71
 1301.33   71.39  1378.2    71.5 1383.16      71  1388.3   70.15
#Mann= 3 ,0,0
       0    .035       0  435.19    .018       0  517.26    .035       0
Levee=-1,296.55,71.77281,-1,547.83,71.77087,	341,	340
Bank Sta=435.19,517.26
XS Rating Curve= 0 ,0
Exp/Cntr=0.3,0.1

Type RM Length L Ch R = 1 ,7544.441,136.14,96.57,56.98
XS GIS Cut Line= 6
     1078809.668    1572315.7257    1078755.1603    1572583.9023
    1078732.1978    1572678.9464    1078622.8718     1572729.903
    1078603.9276    1572741.1766    1078396.2822    1573647.3234
#Sta/Elev= 24
       0    72.5   83.37    72.5  143.29      72  273.01   71.53  273.66   71.75
  298.06   71.75  319.07   70.25  410.06    70.2  431.06   68.71  471.06   68.71
  491.13   70.14  492.06   70.14  581.73   70.12   602.7   71.61  627.12   71.61
  628.96      71 1011.28   70.92 1062.13   70.83  1121.6    70.9 1178.29   70.85
  1202.4      71  1318.7      71 1412.49    71.5 1443.74    71.5
#Mann= 3 ,0,0
       0    .035       0  410.06    .018       0  492.06    .035       0
Levee=-1,298.06,71.74581,-1,602.76,71.61491,	341,	340
Bank Sta=410.06,492.06
XS Rating Curve= 0 ,0
Exp/Cntr=0.3,0.1

Type RM Length L Ch R = 1 ,7447.875,123.11,84.42,45.74
XS GIS Cut Line= 4
     1078660.612     1572303.449    1078611.3139    1572552.2751
    1078568.3847    1572803.1983    1078364.2781    1573635.2584
#Sta/Elev= 24
       0   72.48  157.71    72.5  236.85      72  277.37   71.61  299.04   70.09
  308.61   70.09  329.93   68.61  369.98   68.62  390.79   70.09  508.24   70.09
  529.28   71.59  553.73   71.59   555.5      71  667.43      71  816.89   70.84
  924.02   70.85 1023.66   70.66 1052.44    70.7 1070.11   70.58  1085.2   70.59
  1159.5      71 1245.72      71 1296.12   71.28 1364.96    71.5
#Mann= 3 ,0,0
       0    .035       0  308.61    .018       0  390.79    .035       0
Levee=-1,278.06,71.58557,-1,529.34,71.58852,	341,	340
Bank Sta=308.61,390.79
XS Rating Curve= 0 ,0
Exp/Cntr=0.3,0.1

Type RM Length L Ch R = 1 ,7363.454,84.95,119.85,154.72
XS GIS Cut Line= 5
     1078506.095     1572265.349    1078465.0065    1572577.1945
     1078464.185    1572614.5997    1078546.1793     1572698.458
    1078316.2297    1573634.4117
#Sta/Elev= 26
       0      72   99.46      72  135.64   72.08  183.66   72.31   248.2   72.21
  285.92   71.98  314.49   69.93  387.24   69.97  388.18   69.97  408.24   68.54
  448.24   68.54  469.24   70.04  569.16   70.03  590.24   71.53  614.73   71.53
  616.32      71  680.66      71  763.85   70.83   884.7   70.71   959.9   70.72
  1082.7    70.5 1146.02    70.5 1249.41      71 1329.96      71 1405.88   71.16
 1433.03   71.14
#Mann= 3 ,0,0
       0    .035       0  387.24    .018       0  469.24    .035       0
Levee=-1,184.79,72.31,-1,590.23,71.52976,	341,	340
Bank Sta=387.24,469.24
XS Rating Curve= 0 ,0
Exp/Cntr=0.3,0.1

Type RM Length L Ch R = 1 ,7243.609,70.34,105.57,140.83
XS GIS Cut Line= 4
     1078465.455    1572258.3639    1078431.9017    1572573.9409
    1078412.4907    1572827.8406    1078269.2396    1573625.5217
#Sta/Elev= 21
       0      72  149.71      72  175.69   72.12  287.93      72  317.36    69.9
  434.41    69.9  455.37   68.43   495.7   68.42  516.72    69.9  526.57    69.9
  547.57    71.4  571.97    71.4  573.18      71  746.15   70.57  827.44    70.5
 1134.69    70.5 1164.56   70.83  1209.7      71 1375.52      71 1378.08   70.81
 1382.44   70.89
#Mann= 3 ,0,0
       0    .035       0  434.41    .018       0  516.72    .035       0
Levee=-1,175.1,72.12,-1,547.59,71.4004,	341,	340
Bank Sta=434.41,516.72
XS Rating Curve= 0 ,0
Exp/Cntr=0.3,0.1

Type RM Length L Ch R = 1 ,7138.036,148.73,108.24,67.75
XS GIS Cut Line= 6
    1078440.6899    1572253.2839    1078410.0467     1572572.214
    1078402.5898    1572626.6647     1078303.739    1572699.4352
    1078288.2896    1572714.9299    1078224.1545    1573621.0767
#Sta/Elev= 20
       0      72  290.56      72  320.33   69.87  416.11   69.82  437.11   68.32
  477.11   68.32   497.2   69.76  498.11   69.76   581.1   69.74  602.14   71.24
  626.59   71.23  627.94   70.78  704.89    70.5 1215.23    70.5  1228.5   70.65
 1241.25   70.65 1295.63      71 1422.31      71 1425.83    70.5  1428.4   70.01
#Mann= 3 ,0,0
       0    .035       0  416.11    .018       0  498.11    .035       0
Levee=-1,290.25,71.99,-1,602.22,71.23524,	341,	340
Bank Sta=416.11,498.11
XS Rating Curve= 0 ,0
Exp/Cntr=0.3,0.1

Type RM Length L Ch R = 1 ,7029.794,125.27,88.63,51.99
XS GIS Cut Line= 4
    1078259.0796    1572239.3139    1078248.9277    1572576.7524
    1078259.1448    1572775.2182    1078191.1344    1573617.9017
#Sta/Elev= 24
       0   71.59   29.72   71.63  103.45    71.5  153.63    71.5  240.65      72
   295.2      72  327.46    69.7  338.32    69.7  359.36   68.22   399.3   68.22
  420.26    69.7   536.9   69.71  557.97    71.2  582.45    71.2  583.94   70.71
  637.02    70.5 1196.78    70.5 1270.95      71 1357.37      71 1362.04    70.5
 1365.39      70 1372.89    68.5 1375.74      68 1381.74      68
#Mann= 3 ,0,0
       0    .035       0  338.32    .018       0  420.26    .035       0
Levee=-1,294.2,71.99,-1,558.01,71.20392,	341,	340
Bank Sta=338.32,420.26
XS Rating Curve= 0 ,0
Exp/Cntr=0.3,0.1

Type RM Length L Ch R = 1 ,6941.164,78.58,113.31,148.04
XS GIS Cut Line= 6
    1078140.9693    1572227.8839    1078125.4875    1572526.2204
    1078118.7443    1572619.6797    1078212.2914    1572687.2832
    1078230.5045    1572701.5948    1078163.1944    1573616.6317
#Sta/Elev= 29
       0   71.18   43.56   71.07  140.93    71.5  219.06    71.5  287.77      72
  310.04      72  344.53   69.56  425.86   69.58  426.73   69.58  446.86   68.14
  486.86   68.14  507.86   69.64  605.87   69.66  626.97   71.16  651.49   71.16
  653.15   70.61  686.37    70.5 1281.23    70.5 1318.69   70.61 1325.47   70.69
 1340.26    70.5 1348.24    70.5 1355.67   70.63 1365.51   70.61 1412.81      71
 1426.23      71 1433.13      70 1442.11    68.5 1448.53    68.5
#Mann= 3 ,0,0
       0    .035       0  425.86    .018       0  507.86    .035       0
Levee=-1,309.18,71.99,-1,626.99,71.16149,	341,	340
Bank Sta=425.86,507.86
XS Rating Curve= 0 ,0
Exp/Cntr=0.3,0.1

Type RM Length L Ch R = 1 ,6827.856,73.22,109.5,145.78
XS GIS Cut Line= 5
    1078089.5342    1572224.0739    1078072.2662    1572530.7353
    1078091.3989    1572692.3778    1078104.8158    1572829.0109
    1078096.5192    1573614.0916
#Sta/Elev= 30
       0      71   54.07      71  166.58    71.5  245.34    71.5  317.79   71.99
   352.5   69.51  469.92   69.51  490.89   68.03   530.9   68.03  551.91   69.51
  561.72   69.51  582.72   71.01  607.12   71.01  608.66    70.5  824.03   70.29
  838.62    70.5  903.45    70.5  911.13   70.42   973.2    70.5  988.04   70.16
 1023.09   70.42 1096.64   70.32 1177.09   70.38 1216.09    70.5 1341.61    70.5
 1366.45   70.69 1373.55   70.64 1377.74    70.5 1391.08    70.5 1392.33   70.34
#Mann= 3 ,0,0
       0    .035       0  469.92    .018       0  551.91    .035       0
Levee=-1,317.07,71.98,-1,582.81,71.0098,	341,	340
Bank Sta=469.92,551.91
XS Rating Curve= 0 ,0
Exp/Cntr=0.3,0.1

Type RM Length L Ch R = 1 ,6718.354,130.83,93.53,56.23
XS GIS Cut Line= 6
    1078023.5364    1572218.3589    1078045.1515    1572579.2561
    1078058.2498    1572629.2047    1077972.8051    1572714.3585
    1077960.4596    1572730.8049    1078039.1998    1573628.6967
#Sta/Elev= 30
       0   70.88   78.52      71  181.95    71.5  263.13    71.5   326.9   71.94
  361.54   69.47  451.75   69.43  472.77   67.93   512.8   67.93  532.96   69.37
  533.81   69.37     626   69.34  647.09   70.84  671.59   70.84  673.27   70.28
  729.28   70.11  914.95      70  918.16   70.04  933.12   70.61  964.93   70.28
 1040.61      70 1071.76      70 1089.87   70.14 1190.63    70.1 1275.72    70.5
  1381.5    70.5  1401.9    69.8 1409.14   69.65 1422.37    69.6 1455.71   69.99
#Mann= 3 ,0,0
       0    .035       0  451.75    .018       0  533.81    .035       0
Levee=-1,326.31,71.95,-1,647.12,70.84081,	341,	340
Bank Sta=451.75,533.81
XS Rating Curve= 0 ,0
Exp/Cntr=0.3,0.1

Type RM Length L Ch R = 1 ,6624.823,131.59,94.46,57.33
XS GIS Cut Line= 6
    1077850.8161    1572232.1172    1077906.1448    1572554.4187
    1077914.0826    1572610.7491     1077924.109    1572692.1077
    1077943.7248     1572852.662     1077993.903    1573633.3534
#Sta/Elev= 26
       0   70.25  159.41      71  235.22    71.5  341.95    71.5  372.44   69.32
   383.9   69.32  384.65   69.32  405.23   67.84  444.99   67.84  465.88   69.32
  582.12   69.31  603.17   70.81  627.63    70.8  629.35   70.24  708.45   70.01
  876.52      70  897.14    70.5 1032.99      70 1141.36      70 1212.72    70.3
 1242.65    70.5 1353.36    70.5 1360.11   70.42 1372.04      70 1397.87      70
 1409.93   70.15
#Mann= 3 ,0,0
       0    .035       0   383.9    .018       0  465.88    .035       0
Levee=-1,340.79,71.5,-1,603.18,70.80541,	341,	340
Bank Sta=383.9,465.88
XS Rating Curve= 0 ,0
Exp/Cntr=0.3,0.1

Type RM Length L Ch R = 1 ,6530.362,79.99,110.99,142
XS GIS Cut Line= 6
    1077700.1091    1572245.6639    1077774.2871    1572583.9064
    1077790.7026    1572674.0781    1077886.8148    1572731.9604
    1077901.6162    1572740.9649    1077953.2629      1573641.82
#Sta/Elev= 28
       0      70  140.37      71  183.49    71.5  261.92    71.5  323.27      71
  370.17   70.71  391.74   69.18  467.69    69.2  468.57    69.2  488.81   67.76
  529.02   67.75  550.13   69.25  640.79   69.27  662.05   70.76  686.75   70.76
  688.56   70.16  746.78      70  963.13      70  981.56   70.21 1001.39   70.21
 1057.27      70 1229.18      70 1285.03   70.38 1320.63    70.5 1434.49    70.5
 1441.04   70.41  1451.4    70.5 1469.79    70.5
#Mann= 3 ,0,0
       0    .035       0  467.69    .018       0  550.13    .035       0
Levee=-1,259.61,71.5,-1,662.07,70.76232,	341,	340
Bank Sta=467.69,550.13
XS Rating Curve= 0 ,0
Exp/Cntr=0.3,0.1

Type RM Length L Ch R = 1 ,6419.369,75.69,110.63,145.57
XS GIS Cut Line= 4
     1077636.609    1572260.0573    1077740.8731    1572639.9945
    1077809.3023    1572885.2722    1077905.0028    1573661.2934
#Sta/Elev= 22
       0      70   84.39    70.5  135.63      71  143.89      71  180.44    71.3
  277.11   71.26  360.29   70.63     373   70.63  393.98   69.13  512.11   69.13
  533.12   67.65  573.12   67.65  594.11   69.13   603.2   69.13   624.2   70.63
   648.6   70.63  650.08   70.14  715.95      70 1183.83      70 1277.46   70.41
 1326.95    70.5 1430.53    70.5
#Mann= 3 ,0,0
       0    .035       0  512.11    .018       0  594.11    .035       0
Levee=-1,225.35,71.33,-1,624.23,70.62785,	341,	340
Bank Sta=512.11,594.11
XS Rating Curve= 0 ,0
Exp/Cntr=0.3,0.1

Type RM Length L Ch R = 1 ,6308.738,137.26,95.23,53.18
XS GIS Cut Line= 6
    1077584.9622     1572271.064    1077696.0224    1572605.9842
    1077725.5092    1572696.9381    1077659.7331    1572797.3003
    1077647.6157    1572818.8584    1077849.1227    1573670.6068
#Sta/Elev= 21
       0   69.95   95.65    70.5  170.57   71.02  196.52   71.12  306.69   71.01
  377.18   70.59  398.18   69.09  486.46   69.05  507.46   67.55  547.46   67.55
  567.62   68.99  568.46   68.99   662.1   68.95  683.28   70.45  702.52   70.45
  702.74   70.36     851      70 1301.57      70 1363.22   70.13  1432.3    70.5
 1468.46    70.5
#Mann= 3 ,0,0
       0    .035       0  486.46    .018       0  568.46    .035       0
Levee=-1,197.41,71.12,-1,683.35,70.45068,	341,	340
Bank Sta=486.46,568.46
XS Rating Curve= 0 ,0
Exp/Cntr=0.3,0.1

Type RM Length L Ch R = 1 ,6213.504,134.85,98.46,62.09
XS GIS Cut Line= 5
    1077443.5686    1572310.0107    1077551.8597    1572656.1842
     1077611.188    1572780.7703    1077628.1423    1572851.8785
     1077822.876    1573686.6935
#Sta/Elev= 24
       0   69.78  135.54    70.5  198.52      71   379.1      71  408.15   68.93
  418.07   68.93  439.24   67.46  479.53   67.46  500.71   68.94  618.79   68.92
  640.57   70.45  773.66   70.21  828.17      70 1214.78      70 1230.02   69.87
 1239.88      70 1322.84      70 1354.66   70.15 1368.61    70.5 1373.65    70.5
  1382.9   70.25  1396.7   70.33 1401.82    70.5 1431.04    70.5
#Mann= 3 ,0,0
       0    .035       0  418.07    .018       0  500.71    .035       0
Levee=-1,377.95,71,-1,640.9,70.45,	341,	340
Bank Sta=418.07,500.71
XS Rating Curve= 0 ,0
Exp/Cntr=0.3,0.1

Type RM Length L Ch R = 1 ,6115.049,74.08,109.52,144.96
XS GIS Cut Line= 6
    1077313.1817    1572370.9708    1077423.2416    1572712.0683
     1077468.122    1572801.0784    1077576.7283    1572827.4692
    1077593.4289    1572833.2518    1077788.1626    1573701.9335
#Sta/Elev= 30
       0   70.21   42.98    70.5  123.98    70.5  178.91   70.67  269.18    70.5
  335.65   70.99  373.42   70.95   403.8   68.78  487.87   68.81  508.87   67.37
  548.87   67.37  569.87   68.87  663.35   68.88  687.16   70.55  798.33   70.37
  917.92      70 1230.29      70 1276.75    69.5 1318.59    69.5 1329.36      70
 1392.59      70 1400.07    70.2 1405.43      70 1416.39      70 1432.61    70.5
 1448.72    70.5 1457.27      70 1466.29   68.98 1469.02   68.77 1477.78   68.39
#Mann= 3 ,0,0
       0    .035       0  487.87    .018       0  569.87    .035       0
Levee=-1,373.16,70.95,-1,687.14,70.55,	341,	340
Bank Sta=487.87,569.87
XS Rating Curve= 0 ,0
Exp/Cntr=0.3,0.1

Type RM Length L Ch R = 1 ,6005.533,74.56,110.53,146.5
XS GIS Cut Line= 5
    1077233.9476    1572400.4631    1077387.8418    1572729.4454
    1077445.6147    1572831.2056    1077528.2412    1572994.6647
    1077740.8903    1573719.1491
#Sta/Elev= 19
       0    70.5  172.95    70.5  220.77   70.31  283.52   70.33  380.17   70.77
  408.61   68.74  526.43   68.74  547.49   67.26  587.46   67.26   608.5   68.74
   617.9   68.74  647.39   70.85  695.53    70.5  832.23    70.5   930.4      70
 1333.93      70 1372.57   70.38 1397.81    70.5 1418.42    70.5
#Mann= 3 ,0,0
       0    .035       0  526.43    .018       0   608.5    .035       0
Levee=-1,379.8,70.77,-1,647.29,70.85,	341,	340
Bank Sta=526.43,608.5
XS Rating Curve= 0 ,0
Exp/Cntr=0.3,0.1

Type RM Length L Ch R = 1 ,5895.006,143.8,105.61,67.44
XS GIS Cut Line= 6
    1077188.4392    1572419.5131     1077357.076    1572745.2403
    1077410.6896    1572824.8556    1077363.6318    1572933.3258
    1077354.5979    1572960.3226    1077689.0319    1573749.8408
#Sta/Elev= 23
       0    70.5  151.99    70.5  202.07   70.18  283.61   70.08   345.5    70.5
  385.59   70.61  412.47    68.7  499.01   68.66  520.01   67.16  560.01   67.16
  578.16   68.46  581.01    68.6  677.97   68.57  699.67    70.1  747.63   70.29
  777.85   70.28  833.95      70  929.52      70  953.49    70.2  994.02   70.28
 1069.52      70 1382.95      70 1466.91    70.5
#Mann= 3 ,0,0
       0    .035       0  499.01    .018       0  581.01    .035       0
Levee=-1,385.13,70.61,-1,747.74,70.29,	341,	340
Bank Sta=499.01,581.01
XS Rating Curve= 0 ,0
Exp/Cntr=0.3,0.1

Type RM Length L Ch R = 1 ,5789.398,121.37,83.09,44.79
XS GIS Cut Line= 4
    1077060.3806    1572478.7799    1077233.6889    1572814.6025
    1077383.3932    1573074.5806    1077649.8734    1573773.1242
#Sta/Elev= 29
       0   70.25   22.52   70.24   57.81      70  229.63      70  283.56   69.73
  340.42   69.64  376.94   69.72  377.91   70.04  402.31   70.04  423.31   68.54
  429.95   68.54  451.32   67.06  491.32   67.06  512.44   68.54  632.51   68.54
  653.51   70.04  685.79      70  728.05   70.11  755.84      70  878.72      70
  919.34   70.35  943.87   70.39 1026.02      70 1095.71      70 1123.69   69.79
 1179.03   69.74 1275.93      70  1390.3      70 1425.55   70.17
#Mann= 3 ,0,0
       0    .035       0  429.95    .018       0  512.44    .035       0
Levee=-1,402.31,70.04148,-1,653.5,70.04148,	341,	340
Bank Sta=429.95,512.44
XS Rating Curve= 0 ,0
Exp/Cntr=0.3,0.1

Type RM Length L Ch R = 1 ,5706.307,81.06,119.33,157.59
XS GIS Cut Line= 6
    1076939.7304    1572538.0467    1077111.7443    1572884.8224
    1077159.8641    1572957.1476    1077285.0474    1572971.6098
    1077302.7394    1572979.3726    1077621.2984    1573788.9992
#Sta/Elev= 30
       0      70   40.27      70   66.86    70.5  111.76    70.5  127.91   70.12
  145.57      70   265.4      70  329.82    69.5  385.96    69.5  387.09   69.88
  411.55   69.88  432.59   68.38  517.98   68.43  538.98   66.98  578.98   66.98
  599.98   68.48  697.51    68.5  718.74      70   743.4   69.99  743.84   69.85
  934.84      70 1003.96    70.5 1110.66      70 1157.53      70 1219.69   69.52
 1330.28      70  1452.6      70 1459.15   69.75 1473.79    69.6 1489.35   68.74
#Mann= 3 ,0,0
       0    .035       0  517.98    .018       0  599.98    .035       0
Levee=-1,411.55,69.87965,-1,718.74,69.99842,	341,	340
Bank Sta=517.98,599.98
XS Rating Curve= 0 ,0
Exp/Cntr=0.3,0.1

Type RM Length L Ch R = 1 ,5586.981,78.24,116.23,154.22
XS GIS Cut Line= 5
    1076899.5136    1572560.2718    1077090.7895    1572896.8889
    1077177.9757    1573035.2595     1077246.132    1573153.6204
    1077574.7316    1573815.4576
#Sta/Elev= 30
       0   69.88  120.01    70.5  134.18      70  224.66      70  258.32    69.5
  386.12    69.5  387.17   69.85  411.59   69.85   432.6   68.35  550.71   68.36
  571.73   66.87  611.73   66.87  632.72   68.36   641.9   68.36   662.9   69.86
   687.3   69.86  688.37    69.5  772.12    69.5   872.1      70  923.89      70
  962.03    70.5  991.19    70.5 1123.64    69.5 1251.27      70 1315.92      70
 1323.77    69.5 1333.68   67.96  1348.6    67.5 1376.42      69 1426.22    69.8
#Mann= 3 ,0,0
       0    .035       0  550.71    .018       0  632.72    .035       0
Levee=-1,411.59,69.85081,-1,662.9,69.85725,	341,	340
Bank Sta=550.71,632.72
XS Rating Curve= 0 ,0
Exp/Cntr=0.3,0.1

Type RM Length L Ch R = 1 ,5470.751,132.94,94.95,56.97
XS GIS Cut Line= 6
    1076870.9386    1572577.2051     1077067.716    1572910.1754
    1077118.5891    1572987.8393     1077072.109    1573096.5388
    1077064.6139    1573112.7229    1077505.9398    1573847.2077
#Sta/Elev= 30
       0   69.52   45.93      70  236.11      70   273.2    69.5  385.81    69.5
  386.77   69.82  411.21   69.82  432.24   68.32  515.83   68.26  536.83   66.76
  576.83   66.76  597.83   68.21   696.3    68.2  717.31    69.7  741.71    69.7
  743.77   69.01  749.47   69.01  988.08    69.5  1066.6   69.87 1078.89   69.74
 1097.03   69.19 1138.25    69.5 1206.37    69.5 1379.11      70 1402.13    67.5
 1411.17   67.05 1432.07   68.64  1441.3   69.02 1456.65   69.23 1472.54   68.81
#Mann= 3 ,0,0
       0    .035       0  515.83    .018       0  597.83    .035       0
Levee=-1,411.21,69.82031,-1,717.31,69.70021,	341,	340
Bank Sta=515.83,597.83
XS Rating Curve= 0 ,0
Exp/Cntr=0.3,0.1

Type RM Length L Ch R = 1 ,5375.798,128.33,90.08,51.83
XS GIS Cut Line= 4
    1076754.5217    1572643.8803    1076950.2991    1572977.7881
    1077100.0034    1573237.7662    1077475.2481    1573871.5494
#Sta/Elev= 30
       0    69.5  100.91   69.36  134.67    69.5  181.38    69.2  197.57    69.2
   210.5    69.5  319.08    69.5  385.58   69.16  387.07   69.66  411.47   69.66
  432.47   68.16  441.62   68.16  462.99   66.68     503   66.67  523.77   68.15
  641.67   68.16  662.67   69.66  687.07   69.66  689.05      69  796.94   69.02
 1007.31    69.6 1054.55   69.05 1105.13    69.5 1166.26    69.5 1289.24      70
 1358.44      70 1391.28      67  1397.7      67 1410.88    67.5 1423.61   67.68
#Mann= 3 ,0,0
       0    .035       0  441.62    .018       0  523.77    .035       0
Levee=-1,411.47,69.66111,-1,662.67,69.66111,	341,	340
Bank Sta=441.62,523.77
XS Rating Curve= 0 ,0
Exp/Cntr=0.3,0.1

Type RM Length L Ch R = 1 ,5285.717,76.24,115.71,155.18
XS GIS Cut Line= 6
    1076633.8714    1572711.6137    1076829.4693    1573046.4807
    1076877.2886    1573128.5979    1077000.4639    1573142.8945
    1077024.3972    1573148.7063    1077441.3814    1573888.4828
#Sta/Elev= 28
       0      69   78.73      69  109.78   68.74  166.28    68.5  234.63    68.5
  285.26   68.95  386.39      69  387.88   69.49  412.29    69.5  433.31      68
  524.84   68.04  545.84   66.59  585.84   66.59  606.84   68.09  700.97   68.14
  721.98   69.64  746.38   69.64   748.3      69  762.22   68.99  877.91      69
 1031.25   69.47 1141.26    69.5 1154.27   69.38 1175.95    69.5 1242.76    69.5
 1362.07      70 1473.37      70 1480.67   69.59
#Mann= 3 ,0,0
       0    .035       0  524.84    .018       0  606.84    .035       0
Levee=-1,412.22,69.49541,-1,721.98,69.6356,	341,	340
Bank Sta=524.84,606.84
XS Rating Curve= 0 ,0
Exp/Cntr=0.3,0.1

Type RM Length L Ch R = 1 ,5170.008,86.03,126.37,166.7
XS GIS Cut Line= 5
     1076613.763    1572720.0804    1076806.3819    1573058.7514
    1076892.0198    1573200.3694    1076955.7618    1573319.1616
    1077329.1978    1573958.3329
#Sta/Elev= 30
       0      69   70.07      69  134.95    68.5  246.67    68.5  278.32   68.77
  339.58      69  388.22      69   389.6   69.46  414.06   69.46   435.1   67.96
  555.11   67.97  576.15   66.48  616.17   66.48  637.12   67.97  644.56   67.97
  665.56   69.47  689.96   69.48  692.77   68.54  832.05      69  921.62      69
 1168.96    69.5 1282.43    69.5    1345   69.89 1381.04   69.37 1392.19    69.5
  1403.4      69 1409.36    68.5 1420.71      67 1428.75      67 1430.19   67.18
#Mann= 3 ,0,0
       0    .035       0  555.11    .018       0  637.12    .035       0
Levee=-1,414.06,69.46284,-1,665.53,69.47281,	341,	340
Bank Sta=555.11,637.12
XS Rating Curve= 0 ,0
Exp/Cntr=0.3,0.1

Type RM Length L Ch R = 1 ,5043.642,108.46,72.2,35.89
XS GIS Cut Line= 6
     1076564.143    1572746.4171    1076778.2474    1573072.9603
    1076830.8435    1573143.9279     1076774.338    1573249.5473
    1076768.6134    1573268.3881    1077229.6243    1574017.6896
#Sta/Elev= 30
       0      69   75.71   68.83  114.33    68.5  270.22    68.5  352.44      69
  389.21      69  390.48   69.42  415.29   69.43  436.62   67.93  516.59   67.86
  537.59   66.36  577.59   66.36  598.59   67.83  700.27   67.82  721.48   69.33
  746.11   69.33  748.58   68.52  949.27      69 1035.06      69 1200.76    69.5
  1335.4    69.5 1363.58    68.5 1373.19    66.5 1376.29      66 1387.57      66
 1407.17    68.5 1415.13   69.15 1432.21      70 1468.98    69.5 1498.05    69.5
#Mann= 3 ,0,0
       0    .035       0  516.59    .018       0  598.59    .035       0
Levee=-1,415.26,69.4268,-1,721.41,69.32333,	341,	340
Bank Sta=516.59,598.59
XS Rating Curve= 0 ,0
Exp/Cntr=0.3,0.1

Type RM Length L Ch R = 1 ,4971.438,129.85,93.89,58
XS GIS Cut Line= 4
    1076473.9728    1572787.0572     1076687.982     1573114.152
    1076802.7586    1573391.3524    1077173.7442    1574050.7097
#Sta/Elev= 30
       0    68.5   71.73   68.34  379.43    68.5     389   68.65  390.96    69.3
  415.36    69.3  436.36   67.79  445.03   67.79  466.78   66.29  506.85    66.3
  527.88   67.79  645.56   67.79  666.56   69.29  690.96   69.29  693.32   68.51
  1156.3    69.5 1191.62      70 1212.95      70 1219.94    69.5 1232.91    66.5
 1241.35    65.5 1246.81    65.5 1252.08      66 1257.68   66.73 1266.53    68.5
 1277.26    69.5 1353.11    69.5 1400.12      70 1429.29      70 1447.47   69.66
#Mann= 3 ,0,0
       0    .035       0  445.03    .018       0  527.88    .035       0
Levee=-1,415.32,69.29515,-1,666.51,69.28973,	341,	340
Bank Sta=445.03,527.88
XS Rating Curve= 0 ,0
Exp/Cntr=0.3,0.1
